--- MeadowCrk.prj (project) ---

Proj Title=MeadowCrk
Current Plan=p01
Default Exp/Contr=0,0
English Units
Geom File=g01
Flow File=f01
Plan File=p01
BEGIN DESCRIPTION:
END DESCRIPTION:
DSS Export Rating Curves= 0
DSS Export Rating Curve Sorted= 0
DSS Export Volume Flow Curves= 0
DXF OffsetX= 0
DXF OffsetY= 0
DXF ScaleX= 0
DXF ScaleY= 0

--- MeadowCrk.p01 (plan) ---

Plan Title=Floodplain
Program Version=4.00
Geom File=g01
Flow File=f01
K Sum by GR=0
Std Step Tol=0.01
Critical Tol=0.01
Num of Std Step Trials=20
Max Error Tol=0.3
Flow Tol Ratio=0.001
Split Flow NTrial=30
Split Flow Tol=0.02
Split Flow Ratio=0.02
Log Output Level=0
Friction Slope Method=1
Unsteady Friction Slope Method=2
Unsteady Bridges Friction Slope Method=1
Global Log Level=0
CheckData=False
Run HTab=0
Run UNet=0
Run PostProcess=0
UNET Theta=0
UNET Theta Warmup=0
UNET ZTol=0
UNET ZSATol=0
UNET MxIter=0
UNET MaxInSteps=0
UNET DtIC=0
UNET DtMin=0
UNET MaxCRTS=0
UNET WFStab=0
UNET SFStab=0
UNET WFX=0
UNET SFX=0
UNET DSS MLevel=0
UNET DZMax Abort=0
UNET Convert EG Bridges=0
UNET Use Existing IB Tables=0
UNET Froude Limit=0
UNET Froude Power=0
Write IC File=0
Echo Input=False
Echo Output=False
Write Detailed=0

--- MeadowCrk.f01 (steady flow) ---

Flow Title=NFF Regression Equation
Program Version=4.00
Number of Profiles=1
Profile Names=P100yr
River Rch & RM=MeadowCrk,Main      ,20902.1
426.9552
River Rch & RM=MeadowCrk,Main      ,20609.8
551.0652
River Rch & RM=MeadowCrk,Main      ,18809.8
578.0796
River Rch & RM=MeadowCrk,Main      ,18484.2
756.2840
River Rch & RM=MeadowCrk,Main      ,16377.2
780.2278
River Rch & RM=MeadowCrk,Main      ,15940.1
867.1934
River Rch & RM=MeadowCrk,Main      ,12119.4
949.5938
River Rch & RM=MeadowCrk,Main      ,11862.9
1062.447
River Rch & RM=MeadowCrk,Main      ,11009.8
1099.621
River Rch & RM=MeadowCrk,Main      ,8250.1
1219.039
River Rch & RM=MeadowCrk,Main      ,7509.9
    1500
River Rch & RM=MeadowCrk,Main      ,6753.6
1791.466
River Rch & RM=MeadowCrk,Main      ,209.8
    2200
Boundary for River Rch & Prof#=MeadowCrk,Main      ,1
Up Type=0
Dn Type=3
Dn Slope=0.099997

--- MeadowCrk.g01 (geometry) ---

Geom Title=USGS 3m DEM
Program Version=4.10

River Reach=MeadowCrk       ,Main
Reach XY= 30
     2008161.999      325605.731     2007035.263      323737.675
     2007080.402      322973.787     2007321.722      322918.231
     2007287.486      322402.675     2007755.421      322222.885
     2007602.972      321949.481     2007745.333      321558.856
     2007583.875       321025.87     2007066.513      320421.338
     2006953.666      319996.356     2007067.517      319532.321
     2006846.532      319315.914     2006870.333      319077.953
     2006962.347      318763.717     2007219.638      318553.301
        2007412.      317230.731     2007811.364      316913.431
     2007955.402      316996.356     2008986.652      316437.328
     2009655.564       315577.99     2009895.147      314930.421
     2010384.466      314586.359      2010665.98      313329.726
     2010632.685      313086.402     2010347.945      312814.957
     2009700.702      312534.587     2009651.892      311053.131
     2009334.469      310672.592     2009029.722      309480.784

Type RM Length L Ch R = 1 ,20902.1 ,269.6,292,321
XS GIS Cut Line= 3
     2008462.264      325137.677     2008226.098      325400.957
     2007940.863      326102.754
#Sta/Elev= 30
       0 2752.31    39.3 2737.52    88.4 2721.42   108.1 2716.42     226 2689.09
   245.6 2683.71   265.3 2676.42   304.6 2660.48   353.7 2639.64   413.5 2617.74
   473.3  2594.4   483.3 2591.51   493.2 2590.01   503.2 2589.64   559.8 2590.39
   574.82590.711   582.9 2591.48   602.9 2595.92   612.8    2597   672.6 2598.39
   742.4 2601.02   772.3 2602.88   822.2  2607.1   832.1  2608.5   901.9 2615.35
   971.7  2623.9   981.6 2624.74  1061.4 2633.57  1091.3 2638.03  1111.2 2642.47
#Mann= 3 , 0 , 0
       0      .1       0   559.8    .045       0   574.8      .1       0
Bank Sta=559.8,574.8
XS Rating Curve= 0 ,0
Exp/Cntr=0.3,0.1

Type RM Length L Ch R = 1 ,20609.8 ,285.6,300.1,308.6
XS GIS Cut Line= 3
     2008400.163      325078.891     2007944.406       325403.82
     2007455.171       325648.08
#Sta/Elev= 30
       0 2732.11      20 2723.34      30 2719.27      40 2715.73     110 2695.82
   209.9 2669.02   289.9 2642.25   379.8 2607.93   399.8 2600.98   409.8 2598.57
   429.8 2595.39   552.22579.755   559.7 2579.41   567.22579.792   609.4 2585.16
   619.4    2588   629.3 2592.72   768.5 2668.84   778.4 2673.79   788.4 2677.13
   798.3 2679.14   818.2 2681.65   828.2 2684.08   838.1 2688.81     848 2694.38
   867.9 2704.15   907.7 2720.75   957.4 2743.44  1076.7 2793.79  1106.6 2805.83
#Mann= 3 , 0 , 0
       0      .1       0   552.2    .045       0   567.2      .1       0
Bank Sta=552.2,567.2
XS Rating Curve= 0 ,0
Exp/Cntr=0.3,0.1

Type RM Length L Ch R = 1 ,20309.8 ,313.7,299.8,286
XS GIS Cut Line= 3
     2008360.756      324999.035     2007819.986      325144.917
     2007285.899      325282.143
#Sta/Elev= 30
       0 2728.34      20 2720.32      30 2716.96      40 2714.44      70  2708.1
      80 2705.51     100 2699.35     130 2688.04     170 2670.85     200  2658.8
     300 2621.94   340.1 2608.13   370.1 2598.64   390.1 2593.49   430.1 2585.31
   440.1 2583.66   552.6 2572.08   560.1 2571.57   567.6 2571.79   579.8    2573
   609.3 2577.44   619.2 2579.08     629  2581.7   638.9 2585.38   806.3 2654.16
   904.8 2696.75   993.4  2739.3  1072.2 2779.32  1091.8 2788.48  1111.5 2796.76
#Mann= 3 , 0 , 0
       0      .1       0   552.6    .045       0   567.6      .1       0
Bank Sta=552.6,567.6
XS Rating Curve= 0 ,0
Exp/Cntr=0.3,0.1

Type RM Length L Ch R = 1 ,20009.8 ,289.2,294.7,299.5
XS GIS Cut Line= 3
     2008150.564      324569.524     2007693.456      324892.927
     2007244.583      325199.433
#Sta/Elev= 30
       0  2753.8      70 2719.43     180 2669.71     240 2641.98     260 2634.43
     450 2569.32     460  2567.3     470 2566.27   552.42560.965   559.9 2560.56
   567.42560.674   609.4 2561.97   619.2 2563.04     639 2567.22   648.9 2570.27
   658.8 2574.13   668.6 2578.86   678.5 2584.43   688.4 2590.91   698.3 2597.99
   737.8 2629.58   747.7 2636.97   767.5 2650.32   777.4 2656.16   856.4 2694.93
   905.8 2722.82   955.2  2747.8  1034.3  2783.8  1073.8 2800.72  1103.5 2812.72
#Mann= 3 , 0 , 0
       0      .1       0   552.4    .045       0   567.4      .1       0
Bank Sta=552.4,567.4
XS Rating Curve= 0 ,0
Exp/Cntr=0.3,0.1

Type RM Length L Ch R = 1 ,19715.1 ,312.6,305.2,301.3
XS GIS Cut Line= 3
     2008103.711      324458.367     2007646.185      324589.555
     2007086.603      324878.978
#Sta/Elev= 30
       0 2752.49    39.7 2733.85    89.2 2714.17   257.8 2640.09   287.6  2627.9
     476  2558.9     486 2556.04     496 2554.41     516 2552.34   536.72549.043
     546 2548.29   551.72548.495     586 2551.73     626 2553.22     636  2554.8
     646 2557.77     656 2562.45     666 2568.81     686 2584.24     696 2590.86
     756 2625.58     806 2656.51     816 2661.13     826 2663.54     846 2666.01
     856 2668.79     886 2681.13     946 2708.35    1066 2768.86    1106 2786.36
#Mann= 3 , 0 , 0
       0      .1       0   536.7    .045       0   551.7      .1       0
Bank Sta=536.7,551.7
XS Rating Curve= 0 ,0
Exp/Cntr=0.3,0.1

Type RM Length L Ch R = 1 ,19409.8 ,292.9,300,295.6
XS GIS Cut Line= 3
     2007825.873      324048.651     2007397.346      324386.035
     2006937.286      324685.936
#Sta/Elev= 30
       0  2734.4    49.6 2713.85    79.3 2699.47    99.2 2688.43   128.9  2670.1
   198.3 2630.52   218.2 2624.08   257.8 2615.88   277.7 2609.69   416.5 2548.92
   426.4 2546.09   436.3 2544.83   537.92539.632   552.92539.147   555.4 2539.14
   585.3 2543.79   625.3 2547.67   635.3 2549.37   645.2 2552.56   735.1 2596.87
     835 2655.28     845 2660.96   854.9 2665.13   864.9 2667.59   884.9 2669.88
   934.8 2672.23   944.8 2675.46   954.8 2680.69   994.7 2706.99  1094.6 2765.28
#Mann= 3 , 0 , 0
       0      .1       0   537.9    .045       0   552.9      .1       0
Bank Sta=537.9,552.9
XS Rating Curve= 0 ,0
Exp/Cntr=0.3,0.1

Type RM Length L Ch R = 1 ,19109.8 ,296.1,300,311.2
XS GIS Cut Line= 3
     2007715.204      323876.951     2007227.111      324140.686
     2006804.972       324485.85
#Sta/Elev= 30
       0 2712.38    49.5 2702.87    69.4 2697.41   148.6 2662.51   158.5 2659.01
   168.4 2656.78     208 2651.76   227.9 2646.88   336.8 2606.07   346.7 2601.48
   356.6 2594.84   406.2  2552.2   416.1  2544.9     426 2540.99   547.32528.388
   554.8 2528.04   562.3 2528.29   693.6 2538.19   713.4 2541.42     763 2561.89
   782.8 2571.09   891.9 2628.51   951.4 2657.42   961.3 2661.05   971.2  2663.1
  1020.8 2665.27  1040.6 2667.49  1060.4 2673.85  1070.3 2678.77  1100.1 2697.33
#Mann= 3 , 0 , 0
       0      .1       0   547.3    .045       0   562.3      .1       0
Bank Sta=547.3,562.3
XS Rating Curve= 0 ,0
Exp/Cntr=0.3,0.1

Type RM Length L Ch R = 1 ,18809.8 ,312.1,325.7,341.6
XS GIS Cut Line= 3
     2007638.283      323659.186     2007137.224      323865.504
     2006613.544      324089.017
#Sta/Elev= 30
       0 2701.36    19.7 2695.51      69 2676.68    88.7 2670.62   108.4 2666.32
   118.2 2664.78   147.8  2661.9   167.5  2658.7   206.9 2649.77   226.6 2643.78
   315.3  2608.2     335  2599.6   374.4 2580.06   453.2 2539.12   463.1 2535.82
   472.9 2533.83   502.5 2528.78   522.2 2524.25   534.4 2522.78   541.9 2522.75
   549.4  2523.2   691.7 2528.31   721.7 2529.82   771.6 2533.59   831.6 2540.07
   841.6  2540.7   891.5 2539.74   921.5 2540.83  1031.3 2549.17  1111.3 2559.27
#Mann= 3 , 0 , 0
       0      .1       0   534.4    .045       0   549.4      .1       0
Bank Sta=534.4,549.4
XS Rating Curve= 0 ,0
Exp/Cntr=0.3,0.1

Type RM Length L Ch R = 1 ,18484.2 ,258.7,271.8,283.1
XS GIS Cut Line= 3
     2007617.656      323553.595      2007026.04      323578.886
     2006488.185      323578.886
#Sta/Elev= 30
       0 2687.04   118.4 2662.22   138.2 2656.98   157.9 2648.39   187.5 2630.82
   207.2 2618.16   217.1 2612.48     227 2607.87   256.6 2596.33   296.1 2582.24
   404.6 2546.93   444.1 2530.66   463.9 2523.94   483.6 2519.91   513.2 2516.65
   582.72515.704   592.2 2515.56   597.72515.594     622 2516.76     642 2519.46
   741.6 2540.08   761.5 2545.48   771.4 2549.88   791.4 2560.41   851.1 2593.96
     871 2604.08   920.8 2626.31   990.6 2655.41  1020.4 2665.42    1130  2690.7
#Mann= 3 , 0 , 0
       0      .1       0   582.7    .045       0   597.7      .1       0
Bank Sta=582.7,597.7
XS Rating Curve= 0 ,0
Exp/Cntr=0.3,0.1

Type RM Length L Ch R = 1 ,18212.3 ,279.2,267.3,255.3
XS GIS Cut Line= 3
     2007638.999      323472.005     2007059.111       323309.21
     2006554.677      323266.953
#Sta/Elev= 30
       0 2681.36      79 2656.55    88.9  2652.9    98.7 2647.87   118.5 2634.86
   128.4 2628.88   138.2 2623.87     237 2580.09   246.8 2576.01   256.7 2572.51
   276.5 2566.58   306.1 2559.82   325.8 2556.26   355.5 2552.01   365.3 2549.72
   434.4 2528.95   454.2 2523.74   535.12511.836   543.1 2511.19   550.12511.511
   562.8 2513.14   661.9 2529.02   671.8 2531.85   681.7 2535.77   731.3 2558.11
   761.1  2572.2   870.3 2629.87  1058.9  2723.9  1078.7 2733.13  1108.5 2744.31
#Mann= 3 , 0 , 0
       0      .1       0   535.1    .045       0   550.1      .1       0
Bank Sta=535.1,550.1
XS Rating Curve= 0 ,0
Exp/Cntr=0.3,0.1

Type RM Length L Ch R = 1 ,17945   ,526.8,539.2,551.5
XS GIS Cut Line= 3
     2007660.547      323348.395     2007164.116       323062.21
      2006553.18      323076.102
#Sta/Elev= 30
       0 2679.94    39.5  2669.9    59.3  2663.6      79 2655.75    98.8 2646.61
   118.6 2636.08   138.3  2624.2   187.7  2592.2   217.4 2575.47   237.1 2567.13
   286.5 2551.28   306.3 2546.37   385.3 2529.58   414.9 2523.92   444.6 2519.22
     494 2514.35     573 2509.86   649.92504.091   651.9 2503.96   664.92504.621
   671.6 2505.67   730.7  2522.1   740.6  2525.4   750.4 2529.77   809.6    2560
   878.6 2597.48     987 2652.02  1026.4 2672.41  1075.7 2699.87  1184.1 2762.91
#Mann= 3 , 0 , 0
       0      .1       0   649.9    .045       0   664.9      .1       0
Bank Sta=649.9,664.9
XS Rating Curve= 0 ,0
Exp/Cntr=0.3,0.1

Type RM Length L Ch R = 1 ,17405.6 ,385.2,388.9,391.7
XS GIS Cut Line= 3
     2007867.326      322952.213     2007336.638      322793.651
     2006744.269       322604.94
#Sta/Elev= 30
       0  2699.3    29.7 2688.89    39.6 2684.98   148.4 2638.59     267 2585.54
   326.4 2562.21   474.8 2506.54   484.6 2503.15   494.5 2500.49   504.4 2498.37
   524.2 2494.94   545.7 2490.28   553.9 2489.41   560.72489.542   593.3 2492.08
   662.4  2495.1   711.8 2497.99   731.5 2499.58   741.4 2501.22   780.8 2510.24
   810.4 2514.37   820.3 2516.12   830.2 2518.81   889.4 2539.33   899.3 2543.29
   909.1 2547.86  1027.6  2604.1  1086.8  2633.1  1136.1 2658.38  1175.6 2680.34
#Mann= 3 , 0 , 0
       0      .1       0   545.7    .045       0   560.7      .1       0
Bank Sta=545.7,560.7
XS Rating Curve= 0 ,0
Exp/Cntr=0.3,0.1

Type RM Length L Ch R = 1 ,17016.7 ,275.1,293.6,311
XS GIS Cut Line= 3
     2007885.783      322787.344     2007548.339      322516.602
     2006804.166       322219.99
#Sta/Elev= 30
       0 2641.61   127.8 2583.63     177 2562.42   186.8 2558.89   216.3 2551.85
   245.8 2539.94   255.6 2536.62   275.3 2531.19   324.5 2518.93     413  2494.1
   432.6 2490.18   452.7 2487.85   482.7 2484.98   512.7 2482.87   542.8 2482.15
   652.9 2481.45   709.3 2476.75     723 2475.87   724.32475.923     733 2476.28
   743.1 2479.79   763.1 2490.45   783.1 2498.98   873.2 2528.52   913.3 2543.48
   983.4 2570.94  1053.5 2600.59  1103.6 2622.77  1163.6 2650.19  1233.7 2680.21
#Mann= 3 , 0 , 0
       0      .1       0   709.3    .045       0   724.3      .1       0
Bank Sta=709.3,724.3
XS Rating Curve= 0 ,0
Exp/Cntr=0.3,0.1

Type RM Length L Ch R = 1 ,16722.9 ,383.6,345.7,308.1
XS GIS Cut Line= 3
     2007936.525      322733.285     2007458.548      322208.448
     2007030.175      322141.627
#Sta/Elev= 30
       0 2650.33      50 2631.13      80 2615.92     150 2578.01     200 2554.24
     260 2530.98     270 2527.77     290  2522.6   379.9 2503.44   439.9  2489.9
   519.9  2477.3   529.9 2475.33   549.9 2469.92     5572469.231   559.9 2468.95
     5722469.489   599.9 2474.07   609.9 2475.04   669.9  2478.5   729.6 2480.04
   749.3 2481.24   778.8 2484.62   808.4 2489.95   877.4 2505.18   956.2  2527.5
   966.1 2529.22   985.8 2531.08   995.6 2533.71  1064.6 2560.39  1143.4  2588.4
#Mann= 3 , 0 , 0
       0      .1       0     557    .045       0     572      .1       0
Bank Sta=557,572
XS Rating Curve= 0 ,0
Exp/Cntr=0.3,0.1

Type RM Length L Ch R = 1 ,16377.2 ,420.1,437,453.8
XS GIS Cut Line= 3
     2008239.071      322021.788     2007463.321      322153.559
     2007143.533      322009.177
#Sta/Elev= 30
       0 2514.21    19.9 2510.84    59.8 2506.72    79.7 2503.72    99.6 2498.71
   139.4 2487.03   149.4 2484.71   169.3 2481.59   229.1 2477.71   278.9 2475.67
   398.4 2476.96   438.2 2476.14   468.1 2473.64     508 2465.13   513.52464.802
   517.9 2464.54   528.52464.845     747 2477.16   786.9 2481.14   816.1 2482.88
   835.6 2485.21   933.1 2502.47  1030.5 2523.07    1050 2525.59  1079.2 2525.45
  1098.8 2526.89  1108.5  2529.6  1118.2 2534.28    1128 2541.02  1137.7 2548.68
#Mann= 3 , 0 , 0
       0      .1       0   513.5    .045       0   528.5      .1       0
Bank Sta=513.5,528.5
XS Rating Curve= 0 ,0
Exp/Cntr=0.3,0.1

Type RM Length L Ch R = 1 ,15940.1 ,130.7,120.6,110.4
XS GIS Cut Line= 3
     2008241.531      321900.053     2007435.118      321673.439
     2007147.061      321730.408
#Sta/Elev= 30
       0 2547.49    19.9 2543.22    69.8 2529.89    89.8  2527.1   119.7 2525.12
   139.6 2521.75   179.5  2507.5   219.4 2496.82   239.3  2492.8   259.3 2491.14
   299.2 2490.51   319.1 2486.39     349 2477.14   378.9 2472.76   528.5  2460.2
   544.32459.552   548.5 2459.51   559.3 2459.72   658.2 2462.38   837.6 2470.69
   876.8 2476.48     916 2484.66   984.5 2504.76   994.2 2506.91  1013.8  2508.6
    1053 2514.67  1072.6 2515.68  1111.7 2516.07  1121.5 2516.62  1131.3 2518.74
#Mann= 3 , 0 , 0
       0      .1       0   544.3    .045       0   559.3      .1       0
Bank Sta=544.3,559.3
XS Rating Curve= 0 ,0
Exp/Cntr=0.3,0.1

Type RM Length L Ch R = 1 ,15819.5 ,265.8,251.1,237.6
XS GIS Cut Line= 3
     2008275.089        321641.2     2007740.125      321637.765
     2007123.831      321634.978
#Sta/Elev= 30
       0 2650.39    29.7 2631.63    79.3  2597.9    99.1 2586.65   148.6 2562.37
     208 2537.52   267.5 2518.66   386.4 2479.06     426  2467.5   435.9 2465.26
   445.8 2464.14   475.5 2463.75   485.4 2462.41   505.2 2455.71   515.2 2453.73
   525.1 2453.59   526.6 2453.67   541.62454.614   574.7 2456.81   843.1 2469.07
   892.8 2473.81   912.7 2477.31   942.5 2485.62   972.4 2490.73  1012.1 2501.77
  1101.6 2514.33  1111.5  2517.1  1121.4 2522.15  1141.3 2535.23  1151.3 2540.39
#Mann= 3 , 0 , 0
       0      .1       0   526.6    .045       0   541.6      .1       0
Bank Sta=526.6,541.6
XS Rating Curve= 0 ,0
Exp/Cntr=0.3,0.1

Type RM Length L Ch R = 1 ,15568.4 ,260.3,253.9,248.3
XS GIS Cut Line= 3
     2008173.625      321224.766     2007646.904      321424.331
     2007125.083      321601.407
#Sta/Elev= 30
       0 2512.03    29.6 2507.14    49.4 2501.26    69.2 2493.75      79 2490.68
    88.9 2489.65    98.8 2490.82   138.3 2497.75   148.2 2498.15     168 2495.98
   227.3 2482.21   306.3 2466.95   345.9  2458.5   365.6 2457.04   424.9  2456.2
     5632450.864     578 2450.52   582.9  2450.5   592.8 2450.89   691.2  2459.2
   809.3 2464.36   848.6 2467.91   878.1 2473.39   986.4 2496.76  1006.1  2500.1
  1045.4 2505.56    1075 2511.06  1084.8 2513.47  1094.6 2517.78  1114.3 2531.48
#Mann= 3 , 0 , 0
       0     .06       0     563    .045       0     578      .1       0
Bank Sta=563,578
XS Rating Curve= 0 ,0
Exp/Cntr=0.3,0.1

Type RM Length L Ch R = 1 ,15314.2 ,405,405.4,403.9
XS GIS Cut Line= 3
     2008174.203      320936.844     2007972.148      321008.438
     2007052.709      321431.425
#Sta/Elev= 30
       0    2573    48.7 2559.85   116.9 2539.04   155.9 2527.84   175.4  2520.9
   194.9 2512.41   244.1 2500.91     254 2497.35   273.9 2487.35   293.7  2478.7
   303.7  2475.6   313.6 2473.52   333.4  2470.8   353.3 2469.22   422.7 2468.74
   432.6 2467.91   442.6 2465.64   472.3 2455.74   482.3  2454.5   541.8 2454.51
   643.82449.646   650.9 2449.56   658.82449.615   760.1 2453.36   819.6 2456.23
   839.5 2457.97   988.3 2475.53  1127.2 2491.08  1166.9 2494.97  1226.4 2504.65
#Mann= 3 , 0 , 0
       0     .06       0   643.8    .045       0   658.8     .06       0
Bank Sta=643.8,658.8
XS Rating Curve= 0 ,0
Exp/Cntr=0.3,0.1

Type RM Length L Ch R = 1 ,14908.6 ,294.2,298.7,298.5
XS GIS Cut Line= 3
     2007997.494      320584.053     2007795.439      320690.649
     2006910.404      321176.089
#Sta/Elev= 30
       0 2517.88     9.9  2515.7    29.8 2509.81    39.7  2507.3    59.6 2503.74
   188.7 2489.28   208.6 2486.52   218.5 2484.78   248.4 2478.42   258.4 2475.77
   278.4 2469.12   288.4 2466.66   298.4 2465.42   328.4 2464.14   388.4 2460.66
   448.3 2457.83   508.3 2455.75   578.2 2453.98   690.92449.633   698.2 2449.48
   705.92449.488   898.1 2452.47   908.1 2453.48   918.1 2455.29     978 2467.53
     988 2468.72    1048 2473.78    1078 2476.84  1157.9 2487.38  1237.9 2499.24
#Mann= 3 , 0 , 0
       0     .06       0   690.9    .045       0   705.9     .06       0
Bank Sta=690.9,705.9
XS Rating Curve= 0 ,0
Exp/Cntr=0.3,0.1

Type RM Length L Ch R = 1 ,14609.8 ,327.3,322.9,324.3
XS GIS Cut Line= 3
     2007763.354      320441.097     2007251.383      320650.281
     2006769.786      320917.616
#Sta/Elev= 30
       0 2490.21    29.6 2483.98    59.3 2478.34    69.1 2476.09    98.8 2468.62
   108.6 2466.41   118.5 2464.88   128.4 2463.93     158 2461.84   177.8 2460.18
   187.6  2459.6     316 2454.28   375.3 2452.22   444.4 2450.54   503.7 2450.03
   545.62449.475   553.1 2449.43   560.62449.468   723.3 2450.89   733.3 2451.12
   743.3 2451.62   763.4 2453.34   773.4 2454.39   823.5 2461.09   853.5  2464.6
   883.6 2467.53   953.6 2473.39   973.7 2475.67  1053.8 2485.47  1103.9  2490.7
#Mann= 3 , 0 , 0
       0     .06       0   545.6    .045       0   560.6     .06       0
Bank Sta=545.6,560.6
XS Rating Curve= 0 ,0
Exp/Cntr=0.3,0.1

Type RM Length L Ch R = 1 ,14287   ,266.2,277,286.3
XS GIS Cut Line= 3
     2007581.285      320116.876     2007503.856      320202.662
     2006588.041      320665.514
#Sta/Elev= 30
       0 2477.46    28.9 2477.49    38.5 2476.84    48.2 2475.72    57.8 2474.31
      77 2470.49   115.6 2460.32   125.5 2458.95   145.4  2456.8   165.4 2454.22
   175.3 2453.25   185.3 2452.67     255  2449.4     275 2448.97   354.7 2448.34
   444.3 2448.92   514.1 2448.81   597.22447.902   603.7 2447.83   612.22447.932
     803 2456.29   822.9 2457.64   852.8    2461   872.7 2462.75   892.6 2463.65
   912.6 2464.15   922.5  2464.8    1072 2480.44  1111.8 2485.27  1141.7 2489.48
#Mann= 3 , 0 , 0
       0     .06       0   597.2    .045       0   612.2      .1       0
Bank Sta=597.2,612.2
XS Rating Curve= 0 ,0
Exp/Cntr=0.3,0.1

Type RM Length L Ch R = 1 ,14009.8 ,286.3,299.9,314.6
XS GIS Cut Line= 3
     2007545.359      320010.313     2007026.387      320167.742
      2006475.96      320311.295
#Sta/Elev= 30
       0 2510.85     9.9 2512.23    19.7 2511.75    29.6 2508.96    59.2 2497.01
   118.3 2472.02     138 2464.71   147.9 2461.73   157.8 2459.67   207.1 2452.15
   216.9 2451.31   226.8 2450.98   305.7 2449.65   522.6 2447.72   534.8 2447.72
   549.82447.735   592.2 2448.25     692 2448.74   741.9 2449.82   771.9 2450.93
   801.8 2452.57   851.7 2456.28   861.7 2457.37   891.6 2462.37   931.5 2468.41
   951.5 2472.38  1001.4 2482.94  1021.4 2487.46  1071.2  2500.8  1111.2 2509.99
#Mann= 3 , 0 , 0
       0     .06       0   534.8    .045       0   549.8      .1       0
Bank Sta=534.8,549.8
XS Rating Curve= 0 ,0
Exp/Cntr=0.3,0.1

Type RM Length L Ch R = 1 ,13709.8 ,489.9,473.1,454
XS GIS Cut Line= 3
     2007531.482      319914.704     2006976.236      319893.208
     2006430.818      319837.262
#Sta/Elev= 30
       0 2526.38     9.9  2525.7    19.8 2524.67    29.8 2522.86    39.7 2520.21
   109.2 2495.03   138.9 2483.96   178.6 2469.54   188.5 2466.28   198.4 2463.57
   208.4 2461.36     258 2451.71   267.9 2449.98   277.8 2448.77   287.8  2448.2
   327.4  2447.7   416.8 2447.23   548.22447.712   563.22447.728   695.2 2448.03
   715.2 2448.29     765 2449.62   804.9 2451.51   874.7 2453.96   894.6 2455.21
   984.3 2465.82  1014.2 2468.58  1034.2 2469.64    1074  2470.6  1103.9 2471.87
#Mann= 3 , 0 , 0
       0     .06       0   548.2    .045       0   563.2      .1       0
Bank Sta=548.2,563.2
XS Rating Curve= 0 ,0
Exp/Cntr=0.3,0.1

Type RM Length L Ch R = 1 ,13236.5 ,310.3,319.5,328.4
XS GIS Cut Line= 3
     2007634.582      319270.646     2007090.633       319430.59
     2006376.281      319716.967
#Sta/Elev= 30
       0 2543.35      10  2543.2    19.9 2543.81    39.8 2545.82   129.3 2559.15
   139.3 2560.44   149.2    2561   159.2 2560.42   228.8 2551.73   288.5 2542.61
   318.3 2537.52   358.1  2529.6   387.9 2522.59   407.8 2516.54   437.7 2506.45
   467.5 2495.18   517.2 2474.08     567 2451.12     577 2447.54     587 2446.21
   625.12447.286   640.12447.543   936.8 2452.26  1086.7 2453.85  1126.7 2454.86
  1146.7 2456.24  1206.7 2462.61  1286.6 2472.66  1316.6 2475.22  1336.6  2476.2
#Mann= 3 , 0 , 0
       0      .1       0   625.1    .045       0   640.1      .1       0
Bank Sta=625.1,640.1
XS Rating Curve= 0 ,0
Exp/Cntr=0.3,0.1

Type RM Length L Ch R = 1 ,12917.1 ,386,406.9,425.6
XS GIS Cut Line= 3
     2007502.248      319138.709     2007125.634       319188.76
     2006129.678      319344.677
#Sta/Elev= 30
       0 2512.44      20 2515.77      70 2526.49     130 2540.52     140 2541.86
     150 2541.57     200 2533.54     230 2527.98     260 2521.47   289.9 2514.26
   329.9 2502.85   409.9 2476.78   429.8 2469.94   469.8 2454.86   489.7 2447.86
   499.7 2445.17   509.7 2443.94   529.6 2443.69     6522445.012     6672445.112
   699.3 2446.02     889 2449.19  1018.7 2453.64  1098.6 2454.51  1118.5  2455.9
  1168.4 2461.19  1238.3 2464.42  1278.2 2466.87  1308.2 2469.18    1388 2479.97
#Mann= 3 , 0 , 0
       0      .1       0     652    .045       0     667      .1       0
Bank Sta=652,667
XS Rating Curve= 0 ,0
Exp/Cntr=0.3,0.1

Type RM Length L Ch R = 1 ,12509.8 ,381.8,390.4,401.2
XS GIS Cut Line= 3
     2007521.121      319056.188     2006937.901      318835.501
      2006430.08      318675.902
#Sta/Elev= 30
       0 2502.32    19.8 2495.94    39.6 2490.38    49.5 2488.78    59.4 2489.02
    69.3 2491.04   108.9 2502.08   138.6 2509.04   188.1 2521.71   217.8  2527.7
   227.7 2528.25   237.6 2527.04   247.4 2524.52   336.5  2497.4   445.4 2463.21
   494.9  2444.9   504.8 2442.97   514.7 2442.39   616.12440.822   623.6 2440.64
   631.12440.823   722.2 2445.04   761.6 2446.15   820.7 2446.04   899.6 2443.87
   909.4 2444.05  1037.6 2457.11  1096.7 2460.59  1116.5 2460.38  1155.9 2455.99
#Mann= 3 , 0 , 0
       0      .1       0   616.1    .045       0   631.1      .1       0
Bank Sta=616.1,631.1
XS Rating Curve= 0 ,0
Exp/Cntr=0.3,0.1

Type RM Length L Ch R = 1 ,12119.4 ,264.6,256.3,248.1
XS GIS Cut Line= 2
     2007580.656      318830.789     2006632.429      318227.806
#Sta/Elev= 30
       0 2510.84    79.6 2487.39   149.2 2469.13   159.1 2467.96     169 2468.52
   188.9 2472.36   198.9 2473.05   208.8 2472.79   238.7 2469.22   248.6 2467.42
   268.5 2461.25   298.3 2449.95   308.3 2448.14   387.8 2441.43   441.82439.227
   447.5 2439.06   456.82439.135     706 2441.94   924.8 2441.78   964.6 2443.21
   984.5 2444.51  1004.4 2446.97  1034.2 2451.64  1054.1 2455.92    1064 2458.77
    1074 2463.41  1083.9 2469.62  1103.8 2483.41  1113.8 2488.22  1123.7 2491.83
#Mann= 3 , 0 , 0
       0     .06       0   441.8    .045       0   456.8      .1       0
#XS Ineff= 2 , 0
                          693.09         2456.89
Permanent Ineff=
       F       F
Bank Sta=441.8,456.8
XS Rating Curve= 0 ,0
Exp/Cntr=0.3,0.1

Type RM Length L Ch R = 1 ,11862.9 ,368.4,354.9,341.3
XS GIS Cut Line= 2
     2007892.925       318600.74     2006738.255      318154.402
#Sta/Elev= 30
       0 2471.93    49.9 2470.31   109.8 2466.37   129.8 2466.03   139.8 2465.48
   149.8 2464.44   229.6 2454.17   249.6 2452.08   269.6 2450.45   309.5  2449.2
   339.4 2447.08   379.4 2445.52   419.3 2443.56   519.1 2440.02     629  2438.7
   694.32438.247   698.8 2438.22   709.32438.417   758.7 2440.99   788.7 2442.05
  1098.2 2441.72  1128.1 2442.31  1138.1 2443.04  1148.1 2444.87  1158.1 2447.74
    1178 2455.02    1198 2463.58    1218 2471.37    1228 2474.47  1237.9 2476.55
#Mann= 3 , 0 , 0
       0      .1       0   694.3    .045       0   709.3      .1       0
Bank Sta=694.3,709.3
XS Rating Curve= 0 ,0
Exp/Cntr=0.3,0.1

Type RM Length L Ch R = 1 ,11507.9 ,191.4,198.1,203
XS GIS Cut Line= 2
     2008089.771      318038.479     2006702.433      317987.567
#Sta/Elev= 30
       0 2472.81    69.9 2463.97    79.9 2463.16   129.8 2460.47   139.8 2459.63
   189.8 2454.97   279.6 2445.57   309.6 2443.12   389.5 2440.38   439.4 2439.54
   639.2 2438.69     809 2438.57   827.62438.323     839 2438.23   842.62438.284
   978.8 2439.82  1038.7 2440.77  1078.7 2440.87  1138.6 2440.55  1158.6 2440.73
  1238.5 2445.22  1248.4    2446  1258.4 2447.69  1268.4 2450.48  1308.4 2463.83
  1338.3 2474.41  1358.3 2480.82  1368.3 2484.84  1378.3 2489.78  1388.3 2495.11
#Mann= 3 , 0 , 0
       0      .1       0   827.6    .045       0   842.6     .08       0
#XS Ineff= 2 , 0
           617.2 2449.07
Permanent Ineff=
       F       F
Bank Sta=827.6,842.6
XS Rating Curve= 0 ,0
Exp/Cntr=0.3,0.1

Type RM Length L Ch R = 1 ,11309.8 ,295.9,299.8,305.6
XS GIS Cut Line= 3
     2008038.859      317971.657      2007282.37       317814.93
     2006596.526      317703.791
#Sta/Elev= 30
       0 2462.65    59.4 2459.38    89.1 2457.26   188.2  2448.2   227.8 2445.17
   247.6 2444.08   287.2 2443.06   386.3 2439.36   406.1 2438.98   604.2 2437.86
     723 2437.78   765.12436.843   772.6 2436.76   780.12436.775   881.7 2437.22
   951.2 2437.85  1020.7 2438.82  1040.5  2439.5  1189.4 2448.92  1258.9  2452.8
  1268.8 2453.72  1278.8 2455.25  1298.6 2459.57  1328.4 2465.59  1358.2 2473.65
  1368.1 2475.68    1378 2476.83  1387.9 2477.43  1407.8 2477.54  1467.3 2474.88
#Mann= 3 , 0 , 0
       0     .06       0   765.1    .045       0   780.1     .06       0
Bank Sta=765.1,780.1
XS Rating Curve= 0 ,0
Exp/Cntr=0.3,0.1

Type RM Length L Ch R = 1 ,11009.8 ,594.6,620.2,645.5
XS GIS Cut Line= 3
     2008229.777       317798.24     2007336.769       317523.65
      2006486.07      317261.968
#Sta/Elev= 30
       0 2452.35    29.8 2451.75    99.4 2451.25   129.2  2450.6   178.9 2448.15
   258.4 2442.89   278.3 2441.84   298.2 2441.09   367.8  2439.4   427.4 2437.22
     497 2435.97   596.3 2435.32   785.2 2435.45   926.82436.258   941.82436.407
  1004.3 2437.36  1034.3  2437.5  1094.3  2436.5  1134.3 2435.43  1184.3  2436.7
  1254.3 2439.43  1304.3    2441  1464.3 2442.86  1494.3 2443.53  1524.3 2444.72
  1584.3  2448.6  1634.3 2453.65  1664.3 2454.47  1734.3 2459.81  1824.3 2464.36
#Mann= 3 , 0 , 0
       0     .06       0   926.8    .045       0   941.8     .06       0
Bank Sta=926.8,941.8
XS Rating Curve= 0 ,0
Exp/Cntr=0.3,0.1

Type RM Length L Ch R = 1 ,10389.6 ,568.4,594.4,591.1
XS GIS Cut Line= 2
     2008170.911      317745.737     2007088.626      316344.502
#Sta/Elev= 30
       0 2450.35      90 2446.56     150 2442.33   190.1 2440.79   230.1 2441.09
   270.1  2440.9   290.1 2441.15   330.1 2440.01   380.1 2437.18   410.1 2436.07
   430.1 2435.63   500.2 2435.48   550.2 2434.88   630.2 2434.52   800.92434.732
   815.92434.811   980.3 2436.87  1100.3 2437.94  1210.4 2439.29  1250.4 2440.54
  1390.4 2446.33  1400.4  2447.6  1410.4 2449.99  1450.4 2463.63  1460.4 2466.01
  1590.5 2480.96  1660.5 2490.46  1670.5  2492.1  1690.5  2497.1  1770.5 2518.76
#Mann= 3 , 0 , 0
       0     .06       0   800.9    .045       0   815.9     .06       0
#XS Ineff= 2 , 0
          473.12 2451.81
Permanent Ineff=
       F       F
Bank Sta=800.9,815.9
XS Rating Curve= 0 ,0
Exp/Cntr=0.3,0.1

Type RM Length L Ch R = 1 ,9795    ,229,236.5,245.1
XS GIS Cut Line= 3
     2008479.562      317464.133     2007712.708      316476.132
     2007507.471       316262.94
#Sta/Elev= 30
       0 2472.36      90 2449.41     100 2447.19   110.1 2445.51   140.1 2442.23
   170.1 2438.07   210.1 2434.32   270.2 2431.66   300.2 2430.98   320.2 2430.88
   340.2 2430.95   370.2 2431.44   440.2 2433.46   510.3 2434.64   540.3  2434.9
   640.4  2434.4   743.52432.981   758.52432.989   920.5 2435.78   950.5 2435.95
  1050.6  2437.3  1090.6 2438.54  1160.6 2442.07  1190.6 2442.96  1230.7 2443.07
    1300 2442.49  1319.7 2443.45  1418.4 2449.42  1457.8 2451.18  1546.6 2458.33
#Mann= 3 , 0 , 0
       0     .06       0   743.5    .045       0   758.5     .06       0
Bank Sta=743.5,758.5
XS Rating Curve= 0 ,0
Exp/Cntr=0.3,0.1

Type RM Length L Ch R = 1 ,9558.7  ,335.7,341.3,345.5
XS GIS Cut Line= 2
     2008506.609      317376.629     2007884.534      316044.975
#Sta/Elev= 30
       0 2456.05      20 2450.91      30 2448.91      40 2447.69     120 2440.64
     200 2435.88     230 2434.46     250 2433.88     280 2433.76     370 2433.91
   569.9 2432.57   636.92431.932   639.9 2431.92   651.92432.058   739.9 2434.41
   789.9 2435.29   819.9 2435.54   929.9 2435.45   949.9 2435.58   989.9 2436.26
  1019.8 2437.47  1029.8 2438.08  1059.8 2440.52  1069.8 2441.11  1089.8 2441.98
  1099.8 2442.12  1179.8 2442.27  1269.8 2442.98  1439.8 2442.12  1469.8  2442.2
#Mann= 3 , 0 , 0
       0     .06       0   636.9    .045       0   651.9     .06       0
#XS Ineff= 2 , 0
                          793.86         2439.49
Permanent Ineff=
       F       F
Bank Sta=636.9,651.9
XS Rating Curve= 0 ,0
Exp/Cntr=0.3,0.1

Type RM Length L Ch R = 1 ,9217.1  ,295.2,296.5,296.4
XS GIS Cut Line= 2
     2008715.028      317198.439     2008182.048      315855.648
#Sta/Elev= 30
       0 2451.44    39.8 2448.67    69.7 2446.17    79.7 2445.12   109.6 2440.91
   119.6 2439.82   139.5 2438.72   199.3 2436.46   239.1 2435.52     279 2435.22
   428.4 2436.05   458.3 2436.02   498.2 2435.58     548 2434.55   577.9 2433.14
   608.32431.333   617.7 2431.02   623.32431.042   797.1 2434.05   896.7 2436.58
   996.3 2439.65  1036.2 2440.48  1105.9 2440.97  1145.8 2441.84  1175.7 2442.82
    1365 2450.51  1384.9 2451.68  1394.9  2452.9  1404.8 2454.59  1444.7 2462.49
#Mann= 3 , 0 , 0
       0     .06       0   608.3    .045       0   623.3     .06       0
Bank Sta=608.3,623.3
XS Rating Curve= 0 ,0
Exp/Cntr=0.3,0.1

Type RM Length L Ch R = 1 ,8920.6  ,683.7,670.5,657.6
XS GIS Cut Line= 3
     2009072.999      317381.932     2008764.348      316525.453
     2008442.969       315729.43
#Sta/Elev= 30
       0 2447.31      40  2446.3     110 2443.48   150.1 2442.55   360.2 2440.03
   420.2 2438.59   480.2  2437.7   530.2 2435.52   560.2  2434.8   750.3  2433.5
   840.4 2432.03   870.4 2431.47   899.7 2429.58   910.4 2429.51   914.72429.867
   930.4 2431.07   940.3 2431.36  1229.8 2435.07  1559.2 2441.58  1569.2 2442.24
  1599.2  2445.2  1619.1 2447.28  1629.1 2448.71  1639.1 2451.03    1659 2457.17
    1669  2459.7    1709 2466.41  1718.9 2468.99  1748.9 2478.84  1768.8 2484.64
#Mann= 3 , 0 , 0
       0     .06       0   899.7    .045       0   914.7     .06       0
Bank Sta=899.7,914.7
XS Rating Curve= 0 ,0
Exp/Cntr=0.3,0.1

Type RM Length L Ch R = 1 ,8250.1  ,758.1,739,721.2
XS GIS Cut Line= 4
     2009565.515      317083.147     2009492.845      316420.461
     2008965.267      315790.305     2008956.872       315509.07
#Sta/Elev= 30
       0 2452.39    59.7 2448.36    99.5 2444.77   109.4 2443.58   139.3 2438.26
   149.2 2437.57     408 2434.87   666.7 2434.92   745.9 2433.53   924.1 2433.14
   993.4 2432.06  1052.8 2430.41  1092.4  2428.7  1112.2 2428.38  1116.72428.407
  1128.72428.567  1201.4 2428.93  1330.1 2428.64  1389.5 2428.94  1419.2 2429.76
  1448.9 2430.98  1507.9 2434.52  1614.6 2444.71  1624.3 2446.99    1634 2450.61
  1653.4 2459.05  1663.2 2462.28  1672.8 2464.58  1692.2 2468.28  1769.9 2482.16
#Mann= 3 , 0 , 0
       0      .1       0  1116.7    .045       0  1128.7      .1       0
Bank Sta=1116.7,1128.7
XS Rating Curve= 0 ,0
Exp/Cntr=0.3,0.1

Type RM Length L Ch R = 1 ,7509.9  ,751.4,755.8,759.4
BEGIN DESCRIPTION:
Rating curved added at 8322.3 to correspond with effective WSEL at XS-M.  Channel invert was dropped to correspond to effective profile to allow rating curve to work
END DESCRIPTION:
XS GIS Cut Line= 5
     2011719.028      316154.187     2011035.431      315633.689
      2010168.14      315799.159     2009600.406      315525.278
     2009088.304      315247.117
#Sta/Elev= 30
       0  2457.8     119 2455.41   168.5 2456.26   218.1  2454.1   267.7 2454.87
     347 2450.85   475.9 2456.08   604.8 2451.99     694 2455.87   743.6 2456.41
   862.6    2449     942 2446.39  1090.8 2448.41    1190 2446.98  1328.9 2447.67
  1418.1 2449.39  1547.1 2455.63  1596.7 2454.56  1676.1 2450.18  1746.1 2439.88
  1896.2 2433.26  2016.3 2429.62  2226.4 2427.97  2246.4 2427.78  2256.4 2428.01
  2365.7 2431.68  2543.5 2432.96  2632.4 2437.62  2711.4 2439.78  2889.2 2465.67
#Mann= 3 , 0 , 0
       0     .06       0  2226.4    .045       0  2256.4     .06       0
Bank Sta=2226.4,2256.4
XS Rating Curve= 0 ,0
Exp/Cntr=0.3,0.1

Type RM Length L Ch R = 1 ,6753.6  ,493,511.7,530.4
XS GIS Cut Line= 4
     2011979.904      315844.688      2011346.34      315157.874
     2010296.996      315160.211     2009445.937      314635.117
#Sta/Elev= 30
       0 2462.33   109.3  2473.5     149 2473.93   298.1 2464.74   367.7 2454.46
   417.3 2444.06   447.2 2441.59   665.8 2448.23   814.8 2445.44   844.6 2447.63
   884.4 2455.52   944.3 2456.15  1004.2 2454.88  1084.2 2445.02  1134.2 2445.85
  1184.1 2441.19  1274.1 2456.62  1483.9 2457.89  1663.8 2448.46  1773.8 2449.92
  1863.7 2446.55  1923.7 2448.26  2023.6 2441.54  2103.6 2444.76  2253.7 2441.24
  2403.7 2427.34  2435.72430.688  2450.72432.157  2703.7 2447.38  2943.7 2483.48
#Mann= 3 , 0 , 0
       0     .08       0  2435.7    .045       0  2450.7     .08       0
Bank Sta=2435.7,2450.7
XS Rating Curve= 0 ,0
Exp/Cntr=0.3,0.1

Type RM Length L Ch R = 1 ,6241.6  ,328.6,315.2,287.1
XS GIS Cut Line= 3
     2010598.368      315079.046     2010118.099      314315.222
     2009736.263      314207.035
#Sta/Elev= 30
       0 2451.64    39.7 2452.35   128.9 2456.12   148.7 2455.16   188.4 2449.42
   208.2 2447.94   267.7 2448.32   307.4 2446.68   366.9 2445.95   386.7 2443.44
   426.4 2436.11   446.2 2433.32   475.9 2430.38   525.92427.512   535.4 2427.33
   540.92427.691   565.2 2429.37   624.6 2430.07   674.2 2432.48     694 2436.02
   743.6 2449.76   763.5 2454.12     813 2458.09   832.9 2458.65   902.3 2457.72
   971.7 2452.83  1011.4 2452.04  1110.6 2461.66  1229.7 2466.44  1299.1 2471.92
#Mann= 3 , 0 , 0
       0     .08       0   525.9    .045       0   540.9     .08       0
Bank Sta=525.9,540.9
XS Rating Curve= 0 ,0
Exp/Cntr=0.3,0.1

Type RM Length L Ch R = 1 ,5925.5  ,352.2,323.8,295.3
XS GIS Cut Line= 3
     2010788.434      314788.275     2010603.879      314610.084
     2009944.187      314067.837
#Sta/Elev= 30
       0 2466.43    78.9  2464.1   118.4 2462.24     148 2460.11   207.2 2457.57
   226.9 2455.55   246.7 2452.53   276.4 2445.84   286.3 2444.17   345.9 2436.22
   405.5 2431.78     475 2428.02   504.8 2426.79   554.4 2426.24   565.62426.315
   574.3 2426.86   580.62428.139   584.2 2428.87   594.2 2432.42   623.9 2443.77
   633.9 2446.86   643.8 2448.68     763 2458.48   772.9 2459.05   802.7 2458.87
   911.9 2455.17   951.6 2455.06   991.3 2456.76    1041 2461.47  1110.5 2463.44
#Mann= 3 , 0 , 0
       0     .06       0   565.6    .045       0   580.6     .06       0
Bank Sta=565.6,580.6
XS Rating Curve= 0 ,0
Exp/Cntr=0.3,0.1

Type RM Length L Ch R = 1 ,5601.7  ,359.7,373.3,385.9
XS GIS Cut Line= 3
     2011092.933      314163.194     2010294.168      314177.337
     2009982.605      313993.362
#Sta/Elev= 30
       0 2446.98    89.9 2445.01   119.8 2444.62   239.7  2443.5   299.6 2443.58
   369.5  2442.1   409.4 2440.55   419.4 2439.79   429.4 2438.63   519.3 2427.03
   529.62425.959   539.2 2425.61   544.62425.815   549.2 2425.99   649.1  2434.3
   768.9 2447.37   798.9 2450.51   808.7 2451.18   818.4 2451.71   867.3 2452.25
   886.9 2452.22   916.2 2451.71     926 2451.81    1014 2453.76  1043.4 2454.63
  1072.7 2454.89  1092.3 2455.89  1121.6 2458.36  1131.4 2458.94  1160.7 2459.56
#Mann= 3 , 0 , 0
       0     .06       0   529.6    .045       0   544.6     .06       0
Bank Sta=529.6,544.6
XS Rating Curve= 0 ,0
Exp/Cntr=0.3,0.1

Type RM Length L Ch R = 1 ,5228.4  ,349,346.2,344.4
XS GIS Cut Line= 2
     2011146.935      313982.176     2010094.764      313683.071
#Sta/Elev= 30
       0 2444.93    89.5  2442.5   129.3 2442.02   208.8 2441.57   248.6 2441.12
   278.4 2440.65     348 2439.19   407.7 2437.02   467.4  2434.4   556.9 2430.01
   606.6  2427.3   636.4 2425.48     6422425.418   646.4 2425.37     6572426.329
   666.3 2427.91   676.2 2429.95     706 2435.48     716 2436.84   725.9 2437.58
   765.7 2439.21   785.6 2440.23   865.1 2445.06   904.9 2447.18   924.8 2448.01
   944.7 2448.65   974.5 2449.29   994.4 2449.52  1014.3 2449.44  1093.9 2447.66
#Mann= 3 , 0 , 0
       0     .06       0     642    .045       0     657     .06       0
Bank Sta=642,657
XS Rating Curve= 0 ,0
Exp/Cntr=0.3,0.1

Type RM Length L Ch R = 1 ,4882.1  ,499.9,449.4,399
XS GIS Cut Line= 2
     2011390.019       313678.24     2010349.477      313410.235
#Sta/Elev= 30
       0 2451.61    39.8 2447.88    59.7 2446.32    79.6 2445.21   109.4 2444.03
   139.3 2443.17     189 2442.14   238.8 2440.75   288.5  2439.9   338.3 2439.38
   348.2 2438.92   378.1 2436.19     388  2435.6     398  2435.7   417.9  2436.7
   427.8 2436.65   477.6 2435.04     587  2432.6   626.8 2431.33   779.12425.461
     786 2425.42   794.12425.813   855.6 2431.66   915.3 2436.69   935.2    2438
   955.1 2439.02  1034.7 2441.92  1054.6 2442.16  1064.6 2441.94  1074.5 2441.45
#Mann= 3 , 0 , 0
       0     .06       0   779.1    .045       0   794.1     .08       0
Bank Sta=779.1,794.1
XS Rating Curve= 0 ,0
Exp/Cntr=0.3,0.1

Type RM Length L Ch R = 1 ,4432.6  ,308.9,322.1,326.8
XS GIS Cut Line= 3
     2010884.765      312613.973     2010432.583      313322.448
     2009977.562      313446.545
#Sta/Elev= 30
       0 2445.09      80 2438.87   140.1 2437.33   180.1 2435.23   310.2 2436.29
   360.2 2435.83   380.2 2432.57   390.2 2431.54   460.3 2429.03   490.3 2427.39
   521.1 2422.83   530.3 2422.48   536.12423.135   550.3 2425.29   560.3 2426.14
   600.3 2428.26   680.4 2433.82   740.4 2437.09   800.5 2438.44   840.5 2439.95
     870 2439.74   909.3 2438.55  1007.5  2432.6  1056.6 2432.52  1076.3 2433.92
  1135.2 2442.42  1154.9  2444.4  1253.2 2447.84  1282.6 2449.43  1312.1 2451.89
#Mann= 3 , 0 , 0
       0     .06       0   521.1    .045       0   536.1     .06       0
Bank Sta=521.1,536.1
XS Rating Curve= 0 ,0
Exp/Cntr=0.3,0.1

Type RM Length L Ch R = 1 ,4109.8  ,317.7,300.4,292.8
XS GIS Cut Line= 3
     2010834.089      312554.684     2010405.267      312879.013
     2009948.199      313271.363
#Sta/Elev= 30
       0 2448.51    49.8 2447.58   129.4 2447.09   149.4 2447.38   159.3 2446.84
   169.3 2445.37   179.2 2443.21   199.1 2437.62   209.1 2435.52     219 2434.57
   288.7  2432.2   388.3 2429.65   428.1 2429.36   438.1 2428.92     468 2424.42
   477.9 2423.31   530.22420.203   537.7 2419.82   545.22419.958   557.4 2420.95
   577.2 2423.46   616.7 2424.43   804.3 2436.47   843.8 2438.05   922.8 2439.58
   952.4 2441.01     982 2443.77    1061 2452.47  1120.3 2455.56    1140 2456.25
#Mann= 3 , 0 , 0
       0     .06       0   530.2    .045       0   545.2     .06       0
Bank Sta=530.2,545.2
XS Rating Curve= 0 ,0
Exp/Cntr=0.3,0.1

Type RM Length L Ch R = 1 ,3809.8  ,275.3,264.7,252.8
XS GIS Cut Line= 3
     2010406.163       312231.71     2010161.215      312712.775
     2009879.371      313220.534
#Sta/Elev= 30
       0 2438.57      70  2438.3     110 2437.58     160 2434.42     180 2433.96
   309.9 2435.45   339.9 2434.58   369.9 2432.36   429.9 2431.55   439.9 2430.97
   479.9 2426.29   499.8 2425.71   509.8 2424.78   532.3 2419.58   539.8 2418.38
   547.32418.515   569.9 2420.74   589.9    2422     680 2425.59     700 2426.85
   740.1 2431.73   760.1 2436.43   780.1 2440.01   800.2 2442.28   850.2 2446.57
   970.4 2451.96   980.4 2452.92  1010.4 2457.74  1020.4 2458.74  1120.6    2464
#Mann= 3 , 0 , 0
       0     .06       0   532.3    .045       0   547.3     .06       0
Bank Sta=532.3,547.3
XS Rating Curve= 0 ,0
Exp/Cntr=0.3,0.1

Type RM Length L Ch R = 1 ,3544.9  ,296,338.6,381.2
XS GIS Cut Line= 3
     2010323.839      312191.145     2009947.333      312468.089
     2009798.299      313180.696
#Sta/Elev= 30
       0 2439.75    89.5 2438.81   149.2 2436.21     179 2435.75   467.4 2445.15
   477.4 2444.81   487.3 2443.78   497.3 2441.35   507.3 2437.35   527.2 2426.74
   537.2 2423.58   547.2 2422.73     597 2422.51     607 2421.84   646.9  2416.2
   653.82415.972   656.9 2415.87   668.82417.066   706.7 2424.22   776.6 2432.72
   796.5 2435.88   806.5 2439.04   826.4 2447.58   846.4 2451.24   926.2 2457.59
     996 2459.85  1075.7 2465.18  1115.6 2466.11  1165.5 2465.77  1195.4 2467.22
#Mann= 3 , 0 , 0
       0     .06       0   653.8    .045       0   668.8     .06       0
Bank Sta=653.8,668.8
XS Rating Curve= 0 ,0
Exp/Cntr=0.3,0.1

Type RM Length L Ch R = 1 ,3206.3  ,276.1,285.2,294.2
XS GIS Cut Line= 3
     2010273.676      312134.818     2009912.332       312388.54
     2009178.039      312616.665
#Sta/Elev= 30
       0 2438.49    39.2  2437.4    98.1 2437.05   137.4 2438.91   225.7 2445.15
   255.1 2446.54   284.5 2447.42   382.7 2448.17   441.5 2446.95   451.5 2446.21
   461.5 2443.84   511.4 2427.93   521.4 2425.32   531.4 2424.19   561.4 2423.24
   641.2 2417.65   680.72415.313   681.2 2415.29   691.2 2415.74   695.72416.865
   701.2 2418.24   721.1 2425.64   741.1 2431.49   751.1 2433.38     811 2440.02
     821 2440.82     831 2441.14   920.8 2440.69  1090.6    2443  1210.4 2442.04
#Mann= 3 , 0 , 0
       0     .06       0   680.7    .045       0   695.7     .08       0
Bank Sta=680.7,695.7
XS Rating Curve= 0 ,0
Exp/Cntr=0.3,0.1

Type RM Length L Ch R = 1 ,2920.9  ,301.3,311.1,320.5
XS GIS Cut Line= 3
      2010258.43      312055.439     2009841.533      312165.405
     2009127.891      312222.008
#Sta/Elev= 30
       0 2440.97      49 2440.51    88.2 2441.87   137.2 2445.16   186.2 2449.65
   205.8 2450.38     245 2453.81     294 2456.92   333.2 2458.63   362.6 2458.43
   382.2 2457.11   421.4 2453.45   431.2 2451.48   441.1 2446.76     461 2432.44
   470.9 2426.44   480.9 2423.57   510.7 2422.32   600.2 2415.18   603.52415.203
   618.52415.897   659.8 2419.88   689.7 2421.81   719.5 2423.15   759.3 2424.16
   878.6 2425.38   928.3 2427.25     988 2430.92  1047.6 2431.72    1147 2434.16
#Mann= 3 , 0 , 0
       0      .1       0   603.5    .045       0   618.5      .1       0
Bank Sta=603.5,618.5
XS Rating Curve= 0 ,0
Exp/Cntr=0.3,0.1

Type RM Length L Ch R = 1 ,2609.8  ,402.4,388,373.3
XS GIS Cut Line= 3
     2010268.357      311970.786     2009729.431      311879.688
     2009189.981      311793.884
#Sta/Elev= 30
       0 2443.82    99.4 2443.48   119.2 2443.87   178.9 2447.13   258.4 2453.72
   288.2  2455.7   327.9 2456.76   367.7 2455.84   397.5 2453.43   417.4 2451.01
   427.3 2449.25   437.3  2445.2   457.1  2431.7   467.1 2427.88     477 2426.94
     487 2426.67   496.9 2425.48   526.7  2418.3   539.12415.925   546.6 2415.28
   554.12415.553     626 2421.88   695.5  2429.4   715.4 2430.64     775 2433.04
   874.3 2434.25   904.1 2433.67   943.8 2431.31   983.6 2430.64  1092.8 2434.86
#Mann= 3 , 0 , 0
       0      .1       0   539.1    .045       0   554.1     .08       0
Bank Sta=539.1,554.1
XS Rating Curve= 0 ,0
Exp/Cntr=0.3,0.1

Type RM Length L Ch R = 1 ,2222    ,209.3,212,213.3
XS GIS Cut Line= 3
     2010254.592       311396.05     2009717.559      311493.691
     2009182.629      311607.608
#Sta/Elev= 30
       0 2445.64    39.7    2443    49.6 2442.77   109.2 2446.93   138.9 2447.78
   168.7 2447.59   218.3 2446.28   297.7 2447.61   337.4 2446.81   357.3 2445.44
   416.8 2439.77   446.6 2437.98   476.4 2434.34   486.3 2432.63   496.2  2429.4
   506.1 2425.38   516.1 2423.17     526 2422.56   535.9    2421   545.8 2417.98
   556.52415.474   565.7 2414.87   571.52415.032   625.4 2416.42   675.1 2420.39
   734.8 2422.88   893.9 2424.68   973.4 2426.39  1023.2  2428.1  1092.8  2432.2
#Mann= 3 , 0 , 0
       0      .1       0   556.5    .045       0   571.5      .1       0
Bank Sta=556.5,571.5
XS Rating Curve= 0 ,0
Exp/Cntr=0.3,0.1

Type RM Length L Ch R = 1 ,2009.8  ,304.5,299.8,291.6
XS GIS Cut Line= 3
     2010187.893      311224.727     2009633.972      311295.901
     2009098.668      311391.646
#Sta/Elev= 30
       0 2437.98    39.9 2437.52   219.4 2436.47   229.4 2436.73   269.3 2439.95
   279.2 2440.33   309.2 2440.29     349 2439.07     369 2437.92   398.9  2435.7
   468.7 2428.98   478.7 2426.98   498.6  2419.3   508.6 2418.14   518.6 2418.03
   528.6 2417.18     5512413.025   558.5 2412.14     5662411.989   568.4 2411.94
     598 2412.89   657.4 2416.24   706.8 2419.59   795.8  2426.3   845.2    2429
   874.9  2429.9     954 2431.66   993.5 2432.21  1062.7 2432.62  1102.3 2434.43
#Mann= 3 , 0 , 0
       0      .1       0     551    .045       0     566      .1       0
Bank Sta=551,566
XS Rating Curve= 0 ,0
Exp/Cntr=0.3,0.1

Type RM Length L Ch R = 1 ,1709.8  ,374,356.8,344.4
XS GIS Cut Line= 3
       2010159.1      310872.987     2009638.369      310999.633
     2009078.558      311223.848
#Sta/Elev= 30
       0 2433.43    99.2  2430.4   148.9 2426.98   198.5 2424.45   218.3 2423.79
     258 2424.86   327.5 2428.84   337.4 2428.98   347.4 2428.21   367.2 2425.62
   476.4 2410.63   486.3 2409.85   506.1 2409.09     526 2406.28   528.42406.244
   535.9 2406.13   543.42407.001   575.4 2411.45     615 2414.56   644.7 2416.28
   733.6 2419.27   822.6 2423.62   842.4 2423.97     872 2423.06   881.9 2423.32
   911.6 2425.16     961 2425.03   980.8 2425.53  1020.3 2427.34    1139 2433.88
#Mann= 3 , 0 , 0
       0      .1       0   528.4    .045       0   543.4      .1       0
Bank Sta=528.4,543.4
XS Rating Curve= 0 ,0
Exp/Cntr=0.3,0.1

Type RM Length L Ch R = 1 ,1352.9  ,111.6,116.3,121.8
XS GIS Cut Line= 3
     2009803.984      310608.198     2009427.271      310732.091
     2008964.942      311111.825
#Sta/Elev= 30
       0  2429.1    39.7 2429.04    79.3 2429.86    89.2  2429.7    99.1 2428.77
   128.9 2423.01   188.4 2409.24   208.2 2405.55     228 2402.71   257.8 2400.29
   317.2  2398.2   406.5 2390.68   426.5 2388.42   436.4 2387.65   456.4 2388.98
   496.3 2391.32   556.1 2392.66     576 2393.51     596 2395.32   655.8 2401.92
   675.8 2404.48   695.7 2407.68   705.7 2409.92   735.6  2418.4   765.5 2425.34
   815.4 2431.32   845.3 2431.68   885.2 2432.88     945 2432.84   994.8 2434.89
#Mann= 3 , 0 , 0
       0      .1       0   426.5    .045       0   456.4      .1       0
Bank Sta=426.5,456.4
XS Rating Curve= 0 ,-1
Exp/Cntr=0.3,0.1
